--- ArbckleCrk.prj (project) ---

Proj Title=ArbckleCrk
Current Plan=p01
Default Exp/Contr=0,0
English Units
Geom File=g01
Flow File=f01
Plan File=p01
BEGIN DESCRIPTION:
END DESCRIPTION:
DSS Export Rating Curves= 0
DSS Export Rating Curve Sorted= 0
DSS Export Volume Flow Curves= 0
DXF OffsetX= 0
DXF OffsetY= 0
DXF ScaleX= 0
DXF ScaleY= 0

--- ArbckleCrk.p01 (plan) ---

Plan Title=Floodplain
Program Version=4.00
Geom File=g01
Flow File=f01
K Sum by GR=0
Std Step Tol=0.01
Critical Tol=0.01
Num of Std Step Trials=20
Max Error Tol=0.3
Flow Tol Ratio=0.001
Split Flow NTrial=30
Split Flow Tol=0.02
Split Flow Ratio=0.02
Log Output Level=0
Friction Slope Method=1
Unsteady Friction Slope Method=2
Unsteady Bridges Friction Slope Method=1
Global Log Level=0
CheckData=False
Run HTab=0
Run UNet=0
Run PostProcess=0
UNET Theta=0
UNET Theta Warmup=0
UNET ZTol=0
UNET ZSATol=0
UNET MxIter=0
UNET MaxInSteps=0
UNET DtIC=0
UNET DtMin=0
UNET MaxCRTS=0
UNET WFStab=0
UNET SFStab=0
UNET WFX=0
UNET SFX=0
UNET DSS MLevel=0
UNET DZMax Abort=0
UNET Convert EG Bridges=0
UNET Use Existing IB Tables=0
UNET Froude Limit=0
UNET Froude Power=0
Write IC File=0
Echo Input=False
Echo Output=False
Write Detailed=0

--- ArbckleCrk.f01 (steady flow) ---

Flow Title=NFF Regression Equation
Program Version=4.00
Number of Profiles=1
Profile Names=P100yr
River Rch & RM=ArbckleCrk,Main      ,21473.1
673.6811
River Rch & RM=ArbckleCrk,Main      ,20635.4
679.1160
River Rch & RM=ArbckleCrk,Main      ,20280.3
808.3208
River Rch & RM=ArbckleCrk,Main      ,16576.4
876.7048
River Rch & RM=ArbckleCrk,Main      ,16063.9
985.1789
River Rch & RM=ArbckleCrk,Main      ,14659.8
1010.976
River Rch & RM=ArbckleCrk,Main      ,14319.6
1121.952
River Rch & RM=ArbckleCrk,Main      ,13065.3
1153.812
River Rch & RM=ArbckleCrk,Main      ,8563.9
1277.007
River Rch & RM=ArbckleCrk,Main      ,8272
1531.259
River Rch & RM=ArbckleCrk,Main      ,6163.9
1632.190
Boundary for River Rch & Prof#=ArbckleCrk,Main      ,1
Up Type=0
Dn Type=3
Dn Slope=0.041655

--- ArbckleCrk.g01 (geometry) ---

Geom Title=USGS 3m DEM
Program Version=4.10

River Reach=ArbckleCrk      ,Main
Reach XY= 30
      1927623.77      357172.655     1927741.525        356950.6
     1928021.224      356967.258      1927981.39      356565.636
     1928531.334      356536.153     1928610.203      356784.796
     1929175.854      356868.836     1929798.829      356541.921
     1930165.437      355877.516     1930927.177      355349.259
     1931580.367      355422.655      1932757.74      356012.933
     1933997.034      355255.989     1934512.149      355297.655
     1934951.895       355094.53     1935595.992      355070.225
     1936137.659      355436.544      1937146.99      355475.824
     1937339.048      354950.433      1938054.76      354581.509
     1938264.395      354249.044     1939135.923      354186.544
     1939538.701      353389.669     1939972.729      353037.239
     1940069.907      352556.994     1940587.069      352072.464
     1941278.284      351861.891     1942345.992      351124.044
     1943014.395      351028.558     1944167.147      350306.396

Type RM Length L Ch R = 1 ,21473.1 ,841.5,837.6,824.1
XS GIS Cut Line= 3
     1928048.116      357561.813     1927851.876      357280.778
     1927136.676      356938.962
#Sta/Elev= 30
       0 1940.87    88.1 1939.15   195.9 1942.85   254.6 1942.28   274.2 1944.97
   293.8 1945.26   412.1 1940.03   461.7 1935.94   491.4  1932.4   580.6 1918.56
   587.7 1917.99   600.4 1917.76   602.7 1917.81   649.9  1919.1   659.8 1920.77
   679.7 1925.76   689.6 1927.58   699.5 1928.25   758.9 1929.06   778.8 1927.13
   798.6 1923.76   808.5 1923.14   818.4 1924.38   838.2 1928.25   897.6 1942.46
   917.5 1946.06  1006.6 1952.46  1026.5 1952.49  1115.6 1948.89  1135.4 1948.71
#Mann= 3 , 0 , 0
       0      .1       0   587.7    .045       0   602.7      .1       0
Bank Sta=587.7,602.7
XS Rating Curve= 0 ,0
Exp/Cntr=0.3,0.1

Type RM Length L Ch R = 1 ,20635.4 ,332.3,354.8,376.9
XS GIS Cut Line= 6
      1928476.14      357466.981     1928163.262      356802.955
     1927679.575      356633.057      1927374.28      356771.063
     1927190.607      356854.091     1926432.915      356489.029
#Sta/Elev= 30
       0  1950.8    89.3 1953.12   317.4 1949.94   535.7 1944.16     615 1945.93
   664.6 1945.29   822.8  1933.5   989.4 1914.07  1004.4 1913.98  1010.1 1913.97
  1029.8 1915.81  1079.1 1930.95  1098.8 1935.62  1167.8  1940.4  1177.7 1940.15
  1217.1 1934.99  1276.3 1934.19  1404.4 1927.64  1453.6 1927.14  1552.2 1928.38
  1610.5 1932.07  1668.1 1938.07  1783.3 1942.18  1813.4 1941.78  1923.5 1935.62
  2143.8 1935.86  2273.9 1939.66  2414.1 1949.05  2464.2 1947.31  2624.4 1938.34
#Mann= 3 , 0 , 0
       0      .1       0   989.4    .045       0  1004.4      .1       0
Bank Sta=989.4,1004.4
XS Rating Curve= 0 ,0
Exp/Cntr=0.3,0.1

Type RM Length L Ch R = 1 ,20280.3 ,251.3,253.8,256.8
XS GIS Cut Line= 4
     1928424.021      357311.653     1928187.283      356711.253
     1928098.743      356307.422     1927078.559      355772.355
#Sta/Elev= 30
       0 1953.28   347.5 1947.24   486.5 1948.32   625.5 1935.77   714.3 1918.84
   770.2 1914.18   785.2    1914     793 1913.99   822.6 1914.27   832.4 1916.15
   852.1 1931.99   861.9 1937.19   911.2 1947.28   960.4 1950.05  1019.4 1948.53
  1088.9 1953.24  1219.1 1952.23  1239.1  1950.3  1289.2 1941.32  1469.5 1938.77
  1619.8 1945.86    1720 1942.13    1780 1947.36  1820.1 1948.72  1840.2 1947.44
  1900.3  1936.2  1960.4 1936.32  2010.4 1945.45  2120.6 1973.39  2210.8  1979.1
#Mann= 3 , 0 , 0
       0      .1       0   770.2    .045       0   785.2      .1       0
Bank Sta=770.2,785.2
XS Rating Curve= 0 ,0
Exp/Cntr=0.3,0.1

Type RM Length L Ch R = 1 ,20026.5 ,251.5,285.9,319.1
XS GIS Cut Line= 4
     1928461.786      356964.779     1928429.033      356726.416
     1928394.461      356471.676     1928334.416      356233.312
#Sta/Elev= 30
       0 1951.51   134.7 1948.07     154  1945.7   173.2 1942.22   211.7 1932.82
   221.4 1931.41     231    1931   260.4 1932.41   280.2 1932.56   309.8 1931.25
   369.1 1927.43     379 1924.25   388.9 1919.06   399.2 1914.82   408.7 1913.93
   414.2 1915.22   418.6 1916.25   428.5 1919.87   438.4 1922.13   448.2 1922.67
   497.7 1923.18   517.3 1924.55   527.2  1926.2   566.5 1935.53   586.2 1938.36
     596 1939.02   615.7 1939.36   664.8  1938.6     714 1941.85   743.5 1941.96
#Mann= 3 , 0 , 0
       0      .1       0   399.2    .045       0   414.2      .1       0
Bank Sta=399.2,414.2
XS Rating Curve= 0 ,0
Exp/Cntr=0.3,0.1

Type RM Length L Ch R = 1 ,19740.4 ,127.1,109,91
XS GIS Cut Line= 3
     1928458.702      356710.798     1928657.035      356652.572
     1928802.601      356383.275
#Sta/Elev= 30
       0 1934.54    29.5 1937.37    39.4 1937.97    49.2 1937.44    59.1 1934.66
    68.9 1928.79    78.7 1919.49    88.6 1907.36    98.4 1898.13   100.7 1898.07
   108.3 1897.88   115.7 1903.18     128  1911.9   137.8 1916.74   167.3  1927.3
   177.2 1930.59     187 1933.08   196.9 1934.76   206.7 1936.17   236.3 1939.58
     266 1943.35   325.2 1951.68     345 1953.88   394.3 1957.97   443.7 1963.05
   463.4  1964.8   473.3 1965.43   483.2 1965.81   493.1 1966.05   512.8    1966
#Mann= 3 , 0 , 0
       0      .1       0   100.7    .045       0   115.7      .1       0
Bank Sta=100.7,115.7
XS Rating Curve= 0 ,0
Exp/Cntr=0.3,0.1

Type RM Length L Ch R = 1 ,19631.2 ,280.3,269.6,259
XS GIS Cut Line= 3
     1928462.493      357035.591     1928626.254      356740.821
      1928998.66      356125.806
#Sta/Elev= 30
       0 1951.87    79.3  1950.4   168.6 1945.27   188.4 1942.19   208.3 1934.75
   218.2 1929.96   228.1 1924.02     238 1916.58   257.9 1899.45   267.8 1888.69
   277.7 1879.27   286.4 1875.04   287.6 1874.46   297.5 1877.66   301.4 1881.72
   307.4 1887.97   317.4 1900.24   327.3 1910.02   337.2 1917.49   347.2 1923.64
   357.2 1927.92   377.2 1931.68   556.9  1954.2   626.8 1959.32   696.7 1966.26
   716.7 1967.08   806.5 1965.83   976.3 1968.28  1016.2 1966.83  1056.2 1963.61
#Mann= 3 , 0 , 0
       0      .1       0   286.4    .045       0   301.4      .1       0
Bank Sta=286.4,301.4
XS Rating Curve= 0 ,0
Exp/Cntr=0.3,0.1

Type RM Length L Ch R = 1 ,19361.5 ,124.5,124.9,125.2
XS GIS Cut Line= 3
     1928851.878      357347.604     1928872.048      356591.161
     1929038.533      356235.512
#Sta/Elev= 30
       0 1953.64    89.6 1957.26   139.4 1958.03   258.9 1955.66   288.8 1953.21
   298.7 1950.18   308.7 1944.65   368.4  1900.6   378.4 1894.05   388.3 1888.51
   497.8 1835.64   507.8  1832.3   517.8 1830.15     534 1827.98   537.7  1827.6
     549 1828.44   557.6 1831.05   577.5 1838.81   617.3  1850.1   647.2 1860.77
   667.1 1869.94   756.7 1913.98     796 1928.94   854.9 1956.33   864.7 1960.13
   884.3 1965.53   894.2 1967.26   913.8 1969.07   962.9 1970.74  1149.4 1969.68
#Mann= 3 , 0 , 0
       0      .1       0     534    .045       0     549      .1       0
Bank Sta=534,549
XS Rating Curve= 0 ,0
Exp/Cntr=0.3,0.1

Type RM Length L Ch R = 1 ,19236.7 ,176.8,170.1,162.5
XS GIS Cut Line= 2
     1928983.193       356976.91     1928999.569      356602.078
#Sta/Elev= 30
       0 1876.39     9.9 1872.42    19.8 1868.05    39.5 1858.94    59.2 1850.11
      79 1841.89    88.9  1838.1   118.5 1827.44   148.1 1817.39     158 1814.67
     165 1813.92   167.8 1813.62   177.7 1815.18     180 1815.75   187.6 1817.65
   197.5 1819.79   207.3 1821.45   217.2 1822.86   227.1  1824.5     237 1826.75
   246.8 1829.64   256.7 1832.97   276.4  1840.1   296.2  1846.9   306.1 1850.82
     316  1855.7   325.8 1861.36   335.7 1867.51   345.6 1874.03   375.2 1894.81
#Mann= 3 , 0 , 0
       0      .1       0     165    .045       0     180      .1       0
Bank Sta=165,180
XS Rating Curve= 0 ,0
Exp/Cntr=0.3,0.1

Type RM Length L Ch R = 1 ,19066.4 ,308.2,305,302.8
XS GIS Cut Line= 2
      1929203.21      357098.821     1929043.088      356460.152
#Sta/Elev= 30
       0 1913.74    29.9 1882.37    39.9  1873.5    49.9 1866.73    79.8 1854.53
    99.8  1849.8   129.7 1844.99   139.7 1839.73   149.6  1832.3   169.6 1815.01
   189.6 1800.02   209.5 1790.75   229.4 1789.44   229.6 1789.45   244.6 1790.62
   259.4    1795   279.3 1804.92   299.3 1811.24   319.2 1813.14   389.1 1814.56
     399 1816.46     419  1823.9   448.9 1837.88   468.9 1849.06   528.7 1889.09
   588.6 1932.66   618.5 1952.96   638.5 1965.48   648.5 1970.06   658.4 1972.41
#Mann= 3 , 0 , 0
       0      .1       0   229.6    .045       0   244.6      .1       0
Bank Sta=229.6,244.6
XS Rating Curve= 0 ,0
Exp/Cntr=0.3,0.1

Type RM Length L Ch R = 1 ,18761.3 ,276.8,275.5,274.1
XS GIS Cut Line= 3
      1929744.01      357168.603     1929521.634      356993.286
     1929199.794      356220.756
#Sta/Elev= 30
       0 1965.67    29.3 1965.56    97.6 1960.64   126.9 1957.95   146.5 1954.01
     166 1944.18   185.5 1928.87   205.1 1909.39   244.1 1862.28   253.9 1852.07
   263.6 1844.36   303.1 1834.63   352.9  1813.8   382.8 1804.57   482.4 1798.35
   502.4 1795.75   512.3 1792.28   554.6 1771.37   562.1  1769.9   569.6 1771.27
   631.9 1795.77   771.4 1840.08   801.2 1851.88   831.1 1866.09     881 1892.36
   970.6 1945.41  1000.5 1960.91  1010.5 1963.79  1020.4 1964.13  1120.1 1953.81
#Mann= 3 , 0 , 0
       0      .1       0   554.6    .045       0   569.6      .1       0
Bank Sta=554.6,569.6
XS Rating Curve= 0 ,0
Exp/Cntr=0.3,0.1

Type RM Length L Ch R = 1 ,18485.9 ,147,141,135
XS GIS Cut Line= 3
     1929886.138      357088.743     1929547.108      356380.091
     1929327.401      356149.555
#Sta/Elev= 30
       0 1956.95    19.9 1939.89    69.6  1889.5    89.5 1873.45   109.4 1862.19
   188.9 1838.59   258.5 1807.62   278.4 1799.78   288.4 1797.08   318.2 1794.46
   377.9 1794.08   437.5 1787.35   447.5 1785.42   467.4 1778.87   507.1 1763.83
     527  1753.6   539.3 1749.78   546.9 1749.73   554.3  1751.4   606.6  1763.5
   646.4 1774.74   676.2  1784.2     706 1795.43   755.7 1817.65   845.3  1866.5
   875.1 1880.78   984.6 1912.58  1024.4 1921.84  1064.2 1926.27    1104 1923.78
#Mann= 3 , 0 , 0
       0      .1       0   539.3    .045       0   554.3      .1       0
Bank Sta=539.3,554.3
XS Rating Curve= 0 ,0
Exp/Cntr=0.3,0.1

Type RM Length L Ch R = 1 ,18344.7 ,215.7,205.2,194.6
XS GIS Cut Line= 2
     1929912.134       356702.61     1929602.352      356331.417
#Sta/Elev= 30
       0 1799.11    19.7 1796.15    39.5 1792.53    49.3 1790.38    59.2 1787.77
    69.1 1784.74    88.8 1777.65     148 1753.38   157.9 1748.96   167.7 1743.95
   177.6  1738.5   187.5 1734.85   194.2 1734.51   197.3 1734.35   209.2 1736.53
   217.1 1738.31   226.9  1739.9   256.5 1742.84   276.3 1745.29     296 1748.74
   305.9 1750.83   315.7 1753.69   335.5 1761.32   355.2 1769.92   365.1 1774.53
   414.4 1799.91   453.9 1819.49   463.7 1823.87   473.6 1827.35   483.5 1830.47
#Mann= 3 , 0 , 0
       0      .1       0   194.2    .045       0   209.2      .1       0
Bank Sta=194.2,209.2
XS Rating Curve= 0 ,0
Exp/Cntr=0.3,0.1

Type RM Length L Ch R = 1 ,18139.6 ,268.4,275.7,282.8
XS GIS Cut Line= 2
     1930379.353      356590.618     1929363.332      356167.201
#Sta/Elev= 30
       0 1810.71      40 1808.17      60 1805.08      70 1801.92   110.1 1786.15
   150.1 1773.44   220.1 1748.66   280.2 1730.56   340.2 1716.53   350.2 1715.08
   360.2    1715   400.3 1717.62   450.3 1717.65   490.3 1718.84   500.3 1717.66
   520.3 1713.18   547.9 1703.55   560.4 1702.68   562.9 1703.06   580.4 1705.93
   600.4 1711.75   650.4 1738.86   690.4 1764.03   720.5 1779.09   770.5 1801.24
   890.6 1846.55  1000.6 1886.79  1050.7 1907.63  1080.7 1917.02  1100.7 1921.34
#Mann= 3 , 0 , 0
       0      .1       0   547.9    .045       0   562.9      .1       0
Bank Sta=547.9,562.9
XS Rating Curve= 0 ,0
Exp/Cntr=0.3,0.1

Type RM Length L Ch R = 1 ,17863.9 ,198.9,193.7,188.8
XS GIS Cut Line= 3
     1930426.735      356517.657     1930016.668       356158.23
     1929592.373      355795.999
#Sta/Elev= 30
       0 1803.19    49.6 1788.81    89.2 1775.59   148.7 1757.35   267.7 1717.64
   317.3 1698.39   337.1 1691.81     347 1690.31   356.9 1691.27   396.6 1698.31
   416.4 1699.82   446.2 1697.64   485.8 1692.88   515.6 1688.44   537.8 1683.53
   552.8 1682.52   575.2 1682.98   605.1 1681.95     625 1683.01   664.8 1689.21
   684.8 1694.11   734.6 1708.36   794.4 1729.12   824.2 1740.37   854.1 1753.16
   913.9 1780.61   953.7 1796.68   983.6  1806.6  1033.4  1821.3  1103.2 1838.58
#Mann= 3 , 0 , 0
       0      .1       0   537.8    .045       0   552.8      .1       0
Bank Sta=537.8,552.8
XS Rating Curve= 0 ,0
Exp/Cntr=0.3,0.1

Type RM Length L Ch R = 1 ,17670.2 ,335.7,348.5,361.3
XS GIS Cut Line= 2
     1930571.526      356238.165     1929647.185      355745.061
#Sta/Elev= 30
       0 1739.97    49.9  1730.1   109.8  1719.8   179.6 1703.91   229.5 1694.76
   319.3  1672.2   339.2 1671.31     459 1677.77     469    1677   498.9 1668.11
     508 1667.15   508.9 1667.06     523 1668.96   538.8 1672.92   568.7 1677.52
   648.5  1677.6   668.5 1678.49   698.4 1682.43   728.4 1689.86   748.3  1697.4
   768.3 1707.41   798.2 1726.91   858.1 1770.04     878 1781.88     898 1791.51
   917.9 1798.88   947.9 1806.67   967.8 1809.41  1007.7 1812.46  1047.6 1823.11
#Mann= 3 , 0 , 0
       0      .1       0     508    .045       0     523      .1       0
Bank Sta=508,523
XS Rating Curve= 0 ,0
Exp/Cntr=0.3,0.1

Type RM Length L Ch R = 1 ,17321.8 ,362.7,357.7,352.9
XS GIS Cut Line= 3
     1930606.098      356223.608     1930209.432      355515.795
     1930063.866      355437.554
#Sta/Elev= 30
       0 1737.11    80.1 1715.21   120.2 1705.29   160.3 1696.76   240.4 1681.75
   270.5 1674.08   340.6 1659.04   350.6 1658.03   400.7 1658.62   410.7 1658.16
   450.8  1653.7   490.8 1651.88   520.4 1648.04   530.9 1647.83   535.4 1648.26
   540.9 1648.78     571 1655.02     581 1656.38     591 1657.16     611 1657.59
   691.2 1656.78   751.3 1657.17   791.4 1659.04   811.4 1661.69   869.7 1679.07
   889.2 1684.42   908.6 1689.08     928 1692.47   957.2 1696.64   976.6 1698.92
#Mann= 3 , 0 , 0
       0      .1       0   520.4    .045       0   535.4      .1       0
Bank Sta=520.4,535.4
XS Rating Curve= 0 ,0
Exp/Cntr=0.3,0.1

Type RM Length L Ch R = 1 ,16963.9 ,371.8,387.4,402.9
XS GIS Cut Line= 3
     1931024.635      356003.146     1930656.263      355597.684
     1930291.991      355187.919
#Sta/Elev= 30
       0 1716.69      10 1714.24    19.9 1711.15    39.8  1704.2    89.6 1684.04
   109.6 1677.27   129.5 1671.83   169.3 1659.69   189.2 1654.25   219.1 1647.09
     249 1641.37   268.9 1638.54   288.8 1637.07     488 1633.51   517.9 1632.04
   540.3 1629.32   547.8 1628.88   555.3 1629.48   567.8 1631.92   577.7 1634.87
   587.7 1636.98   597.6 1638.41   647.5 1642.27   687.4 1644.05   787.1    1644
   836.9 1645.24   916.6  1646.3   956.5 1645.36   996.4 1643.39  1096.1 1641.32
#Mann= 3 , 0 , 0
       0      .1       0   540.3    .045       0   555.3      .1       0
Bank Sta=540.3,555.3
XS Rating Curve= 0 ,0
Exp/Cntr=0.3,0.1

Type RM Length L Ch R = 1 ,16576.4 ,505.4,512.3,523.4
XS GIS Cut Line= 5
     1930893.742      355780.846     1930947.552       355562.31
     1930931.925      355276.427     1930574.265      355143.442
     1930755.505      354893.048
#Sta/Elev= 30
       0  1636.6    19.6    1635    48.9  1633.8   127.2 1628.79   225.1 1624.13
   343.5 1622.47   373.2 1621.65   392.9 1620.27   422.5 1616.58   431.8 1616.34
   432.4 1616.32   446.8 1617.05   491.6 1622.75   550.5 1623.25   677.7 1626.32
   746.2    1626   814.7 1624.52     893 1625.25   902.9 1623.68   932.8    1624
   982.7 1622.29  1102.4 1621.02  1112.3    1622  1122.3 1624.23  1132.3 1628.15
  1142.2 1633.79  1152.2 1641.34  1182.1    1668  1192.1 1676.35  1202.1 1683.76
#Mann= 3 , 0 , 0
       0      .1       0   431.8    .045       0   446.8      .1       0
Bank Sta=431.8,446.8
XS Rating Curve= 0 ,0
Exp/Cntr=0.3,0.1

Type RM Length L Ch R = 1 ,16063.9 ,292.7,299.6,302.1
XS GIS Cut Line= 4
     1931287.985      355927.818      1931422.18       355371.62
     1931547.308      355096.789      1931324.98      354831.637
#Sta/Elev= 30
       0  1709.4    39.5 1697.87   108.5 1674.49   266.4 1624.77   295.9 1616.86
   325.5  1610.1   345.3 1607.85     434    1602   564.7 1599.55   572.2 1599.48
   579.7 1599.67   659.8 1603.83     728 1605.95   747.5 1607.78   796.2 1615.62
   815.7 1619.74   844.9 1627.27   874.1 1636.39     884 1638.53   913.7 1647.67
   963.1 1658.18   982.9  1662.9   992.8 1666.34  1002.7 1670.61  1042.2 1691.26
  1081.8 1710.38  1111.4 1726.94  1121.3 1731.91  1141.1 1740.46  1220.2 1771.93
#Mann= 3 , 0 , 0
       0      .1       0   564.7    .045       0   579.7      .1       0
Bank Sta=564.7,579.7
XS Rating Curve= 0 ,0
Exp/Cntr=0.3,0.1

Type RM Length L Ch R = 1 ,15763.9 ,305.8,299.8,294.3
XS GIS Cut Line= 3
     1931385.502      355975.349     1931672.457      355513.889
      1931965.17      355024.973
#Sta/Elev= 30
       0 1723.44    88.9  1694.5   128.4  1682.8   177.8 1669.84   187.7 1666.72
   276.6 1631.75     326 1612.88   335.9 1609.69   345.8 1607.57   355.7 1606.63
   474.2 1599.41   535.9 1594.62   543.4 1594.51   550.9 1594.65   683.4 1599.97
   693.4 1599.75   713.4 1596.52   723.4 1596.48   753.4  1600.7   803.3 1603.72
   823.3 1605.94   883.3 1619.42   933.3 1629.72   983.3 1642.72   993.3 1645.83
  1003.3 1649.43  1023.3 1658.32  1043.3 1668.72  1083.2 1691.07  1113.2 1705.54
#Mann= 3 , 0 , 0
       0     .06       0   535.9    .045       0   550.9     .06       0
#XS Ineff= 2 , 0
                          683.34         1599.93
Permanent Ineff=
       F       F
Bank Sta=535.9,550.9
XS Rating Curve= 0 ,0
Exp/Cntr=0.3,0.1

Type RM Length L Ch R = 1 ,15463.9 ,292.3,300,307.6
XS GIS Cut Line= 3
     1931788.926      356123.394      1931951.34      355592.323
     1932112.685      355072.434
#Sta/Elev= 30
       0 1720.66    59.5 1695.79     119 1673.07   188.4 1654.74   297.5 1622.14
   347.1 1608.92   366.9 1605.34   446.3 1597.75   505.8 1593.75   545.4 1588.74
   547.9  1588.8   555.4 1588.98   562.9 1590.38     585 1594.96   614.7 1596.69
   654.3  1596.7     684  1593.3   693.9 1594.77   713.7 1600.24   723.6 1601.79
   753.3  1603.8   773.1 1606.85   822.6 1617.72   862.2 1627.79   901.8 1639.08
   921.6 1646.85   951.2 1661.73  1020.5 1698.71    1070 1722.53  1099.7 1735.86
#Mann= 3 , 0 , 0
       0     .06       0   547.9    .045       0   562.9     .06       0
Bank Sta=547.9,562.9
XS Rating Curve= 0 ,0
Exp/Cntr=0.3,0.1

Type RM Length L Ch R = 1 ,15163.9 ,305.4,300,293.8
XS GIS Cut Line= 3
     1931885.432      356180.052     1932209.969      355740.972
     1932534.506      355301.892
#Sta/Elev= 30
       0 1735.89    29.8 1726.07    59.6 1714.92    89.4 1702.85   178.7 1671.22
   238.2 1647.68     268 1636.49   317.7 1619.16   367.3  1602.8   377.2 1600.11
   387.2 1598.44   476.5 1592.66   496.4 1590.42   538.5  1583.9   553.5 1583.24
   555.9 1583.23   645.3 1583.82   655.2 1584.28   665.1 1586.77     685 1596.37
   694.9 1599.22   704.8 1600.26   774.3  1603.3   784.2 1604.28   794.2 1606.09
   833.9 1616.59   913.3 1640.22  1022.5 1677.79  1062.2 1690.52    1092 1698.12
#Mann= 3 , 0 , 0
       0     .06       0   538.5    .045       0   553.5     .06       0
Bank Sta=538.5,553.5
XS Rating Curve= 0 ,0
Exp/Cntr=0.3,0.1

Type RM Length L Ch R = 1 ,14863.9 ,209,203.9,199.5
XS GIS Cut Line= 3
     1932251.307      356400.923     1932463.675      355893.055
     1932661.393      355379.196
#Sta/Elev= 30
       0 1798.51      50 1768.58    80.1 1749.59   100.1 1738.13   130.1  1722.9
   170.2 1705.99   220.2 1682.86   270.2 1655.05   320.3 1625.42   330.3 1619.83
   340.3 1615.29   360.3 1608.68   420.4  1590.9   440.4 1588.16     543 1578.48
   550.5  1578.4     558 1578.52   640.6 1580.34   650.6 1583.23   670.6 1594.81
   680.6 1598.67   690.6 1599.86   800.8 1600.72   840.8 1603.68   860.8 1606.96
   890.8 1613.98   950.9  1632.3    1001 1645.75    1051 1662.59  1101.1 1682.07
#Mann= 3 , 0 , 0
       0     .06       0     543    .045       0     558     .06       0
Bank Sta=543,558
XS Rating Curve= 0 ,0
Exp/Cntr=0.3,0.1

Type RM Length L Ch R = 1 ,14659.8 ,351.9,340.2,328.6
XS GIS Cut Line= 3
     1932560.316      356483.806     1932691.325      355721.407
     1932743.553      355403.547
#Sta/Elev= 30
       0 1738.69     9.9 1739.15    29.8 1738.03    59.5 1734.54   128.9 1721.82
   138.8 1719.37   148.8 1715.52   188.4 1691.94   277.7 1642.88   337.2 1608.35
   347.1  1603.4     357 1599.64   386.8 1592.16   416.5 1586.37   507.5 1576.88
   522.5 1576.44   525.6 1576.43   634.7 1577.94   644.6 1578.96   654.6 1582.42
   684.3 1601.19   694.2  1605.1   704.2 1607.01   812.6 1614.44   900.5 1617.38
     920 1619.52   978.6  1632.7  1017.6 1642.98  1046.9 1653.68  1095.7 1675.12
#Mann= 3 , 0 , 0
       0     .06       0   507.5    .045       0   522.5     .06       0
Bank Sta=507.5,522.5
XS Rating Curve= 0 ,0
Exp/Cntr=0.3,0.1

Type RM Length L Ch R = 1 ,14319.6 ,346.8,344,341.2
XS GIS Cut Line= 3
     1933140.823      356452.363     1932962.177       355932.42
     1932780.641      355417.884
#Sta/Elev= 30
       0 1661.42      30 1649.06      70 1634.68      80 1632.48     110 1628.25
   209.9 1609.81   229.9 1607.31   429.8 1588.98   499.8 1584.25   529.8  1580.1
   549.8 1575.31   562.3 1572.97   569.6 1572.45   577.3 1572.61   639.1 1574.39
   688.7 1574.23   698.6 1574.81   708.5 1577.29   718.4 1581.98     778  1614.5
   787.9 1618.06   797.8  1619.4   877.2 1618.42   936.7 1618.44   976.4 1622.36
   986.3 1623.95   996.2 1626.59  1006.1 1630.23  1045.8 1647.48  1095.4 1669.91
#Mann= 3 , 0 , 0
       0     .06       0   562.3    .045       0   577.3     .06       0
Bank Sta=562.3,577.3
XS Rating Curve= 0 ,0
Exp/Cntr=0.3,0.1

Type RM Length L Ch R = 1 ,13975.6 ,313.3,311.2,306.8
XS GIS Cut Line= 3
     1933484.657      356274.556     1933324.535      355914.281
     1933021.712      355306.373
#Sta/Elev= 30
       0 1656.51    19.7 1648.08    39.4 1640.66      69 1632.01   256.3 1591.48
     276  1588.9   384.4 1581.13   486.1 1569.24   494.1 1569.01   501.1 1569.15
     604  1572.9   653.9 1572.29   663.9  1572.4   673.9 1573.44   693.9 1580.14
   733.8 1601.96   753.8 1611.98   763.8 1616.05   773.8 1618.19   783.8 1618.03
   823.7 1611.19   853.7 1608.23   863.7 1607.96   873.7 1608.54   883.6 1610.62
   893.6  1614.7   943.6 1639.53  1023.5 1683.36  1043.4 1695.62  1073.4 1716.57
#Mann= 3 , 0 , 0
       0     .06       0   486.1    .045       0   501.1     .06       0
Bank Sta=486.1,501.1
XS Rating Curve= 0 ,0
Exp/Cntr=0.3,0.1

Type RM Length L Ch R = 1 ,13663.9 ,302.2,300.1,296.2
XS GIS Cut Line= 3
     1933815.157      356122.039     1933528.662       355663.61
     1933175.858      355207.878
#Sta/Elev= 30
       0 1611.42      20 1609.14    70.1 1600.82    90.1 1598.15   110.1 1596.19
   180.2 1591.04   240.3 1585.36   280.3 1582.53   340.4 1579.12   410.4 1575.78
   533.1 1569.22   540.6 1568.93   548.1 1568.94   649.9 1571.04   759.2 1571.29
   769.1 1571.57   779.1 1573.08     789 1576.71   818.8 1590.04   828.8 1594.07
   868.5 1608.14   908.2 1621.64   928.1 1628.98     948 1638.49   977.8 1654.74
   987.8 1659.56   997.7 1663.78  1047.4 1683.57  1087.1 1700.08  1116.9 1711.79
#Mann= 3 , 0 , 0
       0     .06       0   533.1    .045       0   548.1     .06       0
Bank Sta=533.1,548.1
XS Rating Curve= 0 ,0
Exp/Cntr=0.3,0.1

Type RM Length L Ch R = 1 ,13363.9 ,290.9,298.4,309.9
XS GIS Cut Line= 3
     1934072.513      355905.195     1933739.303      355472.812
     1933317.941      355085.274
#Sta/Elev= 30
       0 1691.56    29.8 1682.68    79.4 1666.57     258 1602.98   317.6 1582.56
   337.4 1576.72   347.4 1575.06   357.3 1574.42   446.6 1571.01   516.1 1569.48
   538.4 1568.61   545.9 1568.26   553.4 1568.34   585.4  1570.1     615  1570.8
   733.4 1569.77   743.3 1570.27   753.2  1571.7   792.6 1580.78   832.1 1588.71
   881.5 1600.34   891.3 1601.98   911.1  1604.5   930.8 1608.78   950.6 1613.99
   970.3 1619.69  1019.6 1635.32  1059.1 1647.06  1088.8 1655.14  1118.4 1661.91
#Mann= 3 , 0 , 0
       0     .06       0   538.4    .045       0   553.4     .06       0
Bank Sta=538.4,553.4
XS Rating Curve= 0 ,0
Exp/Cntr=0.3,0.1

Type RM Length L Ch R = 1 ,13065.3 ,293.8,301.4,310.5
XS GIS Cut Line= 3
     1934140.936      355863.073     1933883.143      355100.933
     1933641.705      354848.878
#Sta/Elev= 30
       0 1688.63    19.9 1682.14    89.4    1657   129.1 1643.23   278.1 1596.87
   327.8 1580.41   347.6  1574.9   357.6 1573.61   427.1  1569.5   466.8 1568.82
   506.6 1569.14   594.4  1566.8   605.9 1566.77   609.4 1566.85   615.8 1567.01
   635.7 1570.18   645.6 1571.25   675.4 1571.97   685.4 1572.85   695.3 1574.43
   725.1 1580.98   804.6 1601.01   884.3 1618.02   954.1 1633.88   984.1 1640.94
    1004  1646.3    1024  1652.5  1063.8 1665.97  1113.7  1680.3  1153.6  1693.1
#Mann= 3 , 0 , 0
       0     .06       0   594.4    .045       0   609.4     .06       0
Bank Sta=594.4,609.4
XS Rating Curve= 0 ,0
Exp/Cntr=0.3,0.1

Type RM Length L Ch R = 1 ,12763.9 ,303.4,299.7,291.4
XS GIS Cut Line= 3
     1934220.417      355858.034     1934221.034      355315.016
      1934259.64      354753.438
#Sta/Elev= 30
       0 1697.06    19.8 1693.45    29.6 1690.88    39.5 1687.29   108.6 1653.43
   138.2 1639.55     158 1631.96   187.6 1623.85   197.5 1620.54   207.3 1616.34
   217.2 1611.16   256.7 1587.84   266.6 1582.86   276.4  1579.2   286.3 1577.35
     385 1570.08   414.7 1568.96   454.2 1569.07   535.5 1565.89     543 1565.78
   550.5 1565.86   740.5 1572.61   770.2 1574.86   789.9    1578   809.7  1583.6
   868.9 1602.44   947.9 1625.96    1017 1651.69  1066.4 1669.52  1105.9 1684.92
#Mann= 3 , 0 , 0
       0     .06       0   535.5    .045       0   550.5     .06       0
Bank Sta=535.5,550.5
XS Rating Curve= 0 ,0
Exp/Cntr=0.3,0.1

Type RM Length L Ch R = 1 ,12463.9 ,306,300,295.5
XS GIS Cut Line= 3
      1934604.84      355829.914      1934518.28      355296.471
     1934346.986      354745.631
#Sta/Elev= 30
       0    1672      20 1663.41      30 1660.44      40 1659.03      70 1659.07
   170.1 1646.62   200.2 1642.05   210.2 1639.54   250.2  1626.4   280.2 1618.03
   390.3 1575.91   400.3 1572.64   410.3 1570.53   420.3 1569.48   440.3 1568.71
   490.4 1568.65   500.4 1568.17   532.9  1564.9   540.4 1564.62   547.9 1564.64
   739.3 1570.03   828.8 1573.76   848.7 1575.54   858.7 1577.12   878.6  1581.7
   908.4 1589.89   958.2 1606.15     978 1613.26  1027.8 1632.52  1117.3 1672.25
#Mann= 3 , 0 , 0
       0     .06       0   532.9    .045       0   547.9     .06       0
Bank Sta=532.9,547.9
XS Rating Curve= 0 ,0
Exp/Cntr=0.3,0.1

Type RM Length L Ch R = 1 ,12163.9 ,291.4,298.8,308.4
XS GIS Cut Line= 3
     1934998.772       355657.53     1934773.679      355156.565
     1934513.835       354676.13
#Sta/Elev= 30
       0 1656.47    59.9 1651.69    89.9 1648.47   119.8 1644.05   159.8 1636.76
   189.7 1632.39   199.7 1631.56   229.7 1630.88   249.6 1628.25   259.6 1627.37
   279.6 1626.86   289.6 1625.19   299.6  1622.6   319.5 1615.92   329.5 1612.16
   359.5 1599.04   369.5 1595.46   399.4 1587.09   429.4 1580.29   449.4  1576.6
   541.7 1564.39   556.7 1563.68   559.1 1563.65   747.8 1566.91   767.7 1568.66
   807.4  1573.4   817.4 1575.21   936.5 1615.18   976.2  1625.6  1095.4 1662.43
#Mann= 3 , 0 , 0
       0     .06       0   541.7    .045       0   556.7     .06       0
Bank Sta=541.7,556.7
XS Rating Curve= 0 ,0
Exp/Cntr=0.3,0.1

Type RM Length L Ch R = 1 ,11865   ,299.2,301.1,302.7
XS GIS Cut Line= 3
     1935112.081      355628.053     1935059.496      355084.671
     1935027.025      354539.182
#Sta/Elev= 30
       0 1627.51    39.7 1625.36     129 1621.88   158.8 1619.64   198.5 1615.81
   218.4 1613.09   238.2 1609.52   317.6 1589.83   357.3 1582.18   377.2  1579.7
   416.9 1577.45   426.8 1576.44   506.2 1566.94   526.1 1562.86     531  1562.4
   545.9 1561.71     546 1561.71   595.6 1562.67   615.5 1564.44   645.3 1568.06
   655.2 1568.49     695 1567.82   744.6 1568.44     844  1573.4   943.3 1580.32
   983.1 1582.24     993 1583.19  1012.9 1587.21  1072.5 1602.15  1092.4 1608.19
#Mann= 3 , 0 , 0
       0      .1       0     531    .045       0     546      .1       0
#XS Ineff= 2 , 0
                          612.41         1570.18
Permanent Ineff=
       F       F
Bank Sta=531,546
XS Rating Curve= 0 ,0
Exp/Cntr=0.3,0.1

Type RM Length L Ch R = 1 ,11563.9 ,289.8,295.5,300.8
XS GIS Cut Line= 3
     1935365.274       355600.61     1935358.001        355054.6
     1935358.001       354508.61
#Sta/Elev= 30
       0 1694.39    89.4 1667.15   168.8 1641.72   178.7 1639.07   228.4  1627.8
   238.3 1625.08   317.7 1598.83   377.3 1578.44   387.2 1576.33   397.1 1575.28
   496.4 1565.97   506.4 1564.48   526.2 1560.76   538.6 1559.17   546.1 1558.86
   553.6 1559.35   575.8 1561.06   744.6  1571.1     834 1573.72   843.9 1574.76
   853.8 1576.42   893.5 1584.47   903.4 1585.74   913.4  1586.3   982.8 1587.96
  1052.3 1589.02  1062.3  1589.7  1072.2 1590.99  1082.1 1592.92    1092 1595.52
#Mann= 3 , 0 , 0
       0      .1       0   538.6    .045       0   553.6      .1       0
Bank Sta=538.6,553.6
XS Rating Curve= 0 ,0
Exp/Cntr=0.3,0.1

Type RM Length L Ch R = 1 ,11268.3 ,272.6,283.8,292.3
XS GIS Cut Line= 3
     1935453.907      355612.221     1935619.012      355215.566
     1935779.193       354553.16
#Sta/Elev= 30
       0 1698.44      20 1694.22      30 1691.68    79.9 1676.85   129.9 1660.46
   159.9 1648.92   179.8 1641.91   259.8 1617.32   329.7 1594.59   359.7 1585.92
   399.7 1575.14   409.7 1573.24   419.6 1572.12   518.5  1563.7   561.3 1559.43
   567.9 1558.84   576.3  1558.7   577.8 1558.67   587.7  1559.6   597.6 1561.57
   656.8 1575.57   735.8 1596.88     805 1619.12   972.9 1681.38   992.6 1688.13
  1002.5 1690.97  1022.2 1695.67  1061.8 1703.19  1081.5 1706.17  1111.1 1709.79
#Mann= 3 , 0 , 0
       0      .1       0   561.3    .045       0   576.3      .1       0
Bank Sta=561.3,576.3
XS Rating Curve= 0 ,0
Exp/Cntr=0.3,0.1

Type RM Length L Ch R = 1 ,10984.7 ,329.8,320.6,313.2
XS GIS Cut Line= 3
     1935515.125      355641.653     1935902.613      355210.759
     1936207.055      354764.649
#Sta/Elev= 30
       0 1708.15      60 1697.14    79.9  1692.6    89.9 1689.58   119.9 1679.26
   189.8  1653.1   209.8 1646.04   329.7 1605.66   419.6 1577.09   429.6 1574.74
   449.6 1571.83   509.6 1566.68   567.9 1558.91   569.5 1558.72   579.5 1558.76
   582.9 1559.29   589.5 1560.33   649.5  1573.9   689.5 1583.39   709.5 1588.67
   749.5 1601.01   799.5  1618.3   819.5 1624.58   869.6 1637.07   909.6 1649.44
   929.6 1654.95  1029.6 1684.95  1049.6 1691.22  1089.6 1706.01  1119.6 1715.37
#Mann= 3 , 0 , 0
       0      .1       0   567.9    .045       0   582.9      .1       0
Bank Sta=567.9,582.9
XS Rating Curve= 0 ,0
Exp/Cntr=0.3,0.1

Type RM Length L Ch R = 1 ,10663.9 ,331,322.2,313.9
XS GIS Cut Line= 3
     1935947.826      355933.263     1936115.824      355429.266
     1936295.324      354825.872
#Sta/Elev= 30
       0 1757.66   236.1 1659.17   255.8 1652.25   354.2 1621.64   432.9 1591.79
   462.4 1577.85   472.2 1573.87   491.9 1567.74   511.6  1560.7   521.4 1557.86
   523.8 1557.59   531.3 1556.75   538.8 1557.01   561.2 1559.11   631.2 1564.06
   671.2 1565.45   681.2 1566.29   711.1 1570.41   741.1 1576.29     831 1598.19
     871 1609.52     921 1622.52   970.9 1640.55   980.9 1643.46  1000.9 1648.11
  1020.9    1654  1050.9 1664.55  1100.8 1684.07  1130.8 1694.07  1160.8  1702.7
#Mann= 3 , 0 , 0
       0      .1       0   523.8    .045       0   538.8      .1       0
Bank Sta=523.8,538.8
XS Rating Curve= 0 ,0
Exp/Cntr=0.3,0.1

Type RM Length L Ch R = 1 ,10341.7 ,275.5,283,290.7
XS GIS Cut Line= 2
      1936464.69      355948.608     1936375.983      354828.259
#Sta/Elev= 30
       0 1641.04    69.6 1630.66    99.5  1625.5   119.4 1620.66   159.1  1608.1
   198.9 1596.88   218.8 1591.92   238.7 1588.46   278.5 1584.18   308.3 1583.64
   377.9 1574.23   457.5 1566.57     574 1556.46   586.8 1556.13     589 1556.52
   596.7 1557.88   606.7 1562.16   616.6 1567.52   646.5 1580.01   656.4 1583.33
   686.2 1589.14   696.2 1592.14   765.8 1621.59   775.8 1625.31   795.6 1631.56
   934.9 1671.61   974.7 1682.21  1004.5 1689.17  1054.2 1698.35  1123.9 1712.87
#Mann= 3 , 0 , 0
       0      .1       0     574    .045       0     589      .1       0
Bank Sta=574,589
XS Rating Curve= 0 ,0
Exp/Cntr=0.3,0.1

Type RM Length L Ch R = 1 ,10058.7 ,299,292.4,285.9
XS GIS Cut Line= 3
     1936551.981       355953.05     1936705.295       355370.23
       1936650.9      354839.607
#Sta/Elev= 30
       0 1673.52    29.6 1669.15    69.2 1659.97    98.8 1654.59   108.7 1651.62
   138.3 1640.76   227.2  1620.4   237.1 1617.82   266.8 1607.63   276.6 1605.15
   395.2 1579.43   434.7 1571.42   464.3 1566.02   532.2 1555.85   543.4 1555.35
   547.2 1555.73   553.2 1556.34   563.1 1559.24     573 1562.93   632.3 1580.88
   691.6 1602.56   750.8 1621.85   829.8 1649.76   849.6 1655.38   869.4 1661.98
   908.9 1676.33     978 1702.99    1057 1729.56  1076.8 1737.91    1136 1771.21
#Mann= 3 , 0 , 0
       0      .1       0   532.2    .045       0   547.2      .1       0
Bank Sta=532.2,547.2
XS Rating Curve= 0 ,0
Exp/Cntr=0.3,0.1

Type RM Length L Ch R = 1 ,9766.1  ,374.7,347.5,320.2
XS GIS Cut Line= 3
     1936992.616      356002.693     1936972.772      355430.276
     1936729.986      354839.537
#Sta/Elev= 30
       0  1647.3    49.4 1644.52   108.6 1639.75   167.9 1632.34   227.1 1622.53
   266.6 1614.78   325.9  1601.1   385.1  1585.8     474 1561.76   513.4 1554.77
   523.4 1554.31   528.4 1554.51   543.1 1555.87   582.7 1561.18   622.7 1564.46
   642.6 1566.73   662.6 1571.13   702.5 1582.46   852.2 1630.65   892.1 1643.02
     962 1659.63   981.9 1664.92   991.9  1668.4  1041.8 1688.72  1081.7 1703.94
  1101.7 1710.65  1141.6 1722.71  1161.6 1729.64  1191.5 1741.87  1211.4  1751.9
#Mann= 3 , 0 , 0
       0      .1       0   513.4    .045       0   528.4      .1       0
Bank Sta=513.4,528.4
XS Rating Curve= 0 ,0
Exp/Cntr=0.3,0.1

Type RM Length L Ch R = 1 ,9418.5  ,224.5,226.8,229.3
XS GIS Cut Line= 3
     1937705.828      355496.232     1937089.225       355282.89
     1936790.304      354808.323
#Sta/Elev= 30
       0 1619.57    19.8 1621.45    39.5 1622.05   138.4 1618.56   158.2 1617.24
   207.6  1612.2   266.9 1608.66   286.7  1606.4   425.1 1583.55   464.6 1576.12
   474.5 1573.33   484.4 1569.26   494.3 1564.25     524 1546.19   531.2 1544.68
   533.8 1544.14   546.2 1545.39   573.4 1550.88   622.8 1559.38   642.6 1564.37
   692.5 1579.22   712.6 1582.84   722.6 1585.43   882.8 1636.69     993 1665.02
  1093.2 1701.48  1163.2 1722.83  1183.3 1729.84  1193.3  1734.1  1213.3 1744.34
#Mann= 3 , 0 , 0
       0      .1       0   531.2    .045       0   546.2      .1       0
Bank Sta=531.2,546.2
XS Rating Curve= 0 ,0
Exp/Cntr=0.3,0.1

Type RM Length L Ch R = 1 ,9191.5  ,308.9,327.3,345.6
XS GIS Cut Line= 3
     1937720.615      355321.101     1937167.466      355059.083
     1936799.897       354725.67
#Sta/Elev= 30
       0 1600.17    39.5 1601.67    69.1 1601.84   167.8 1598.61   286.3 1591.84
   355.4 1586.36   365.3 1584.48     385 1578.16   434.4 1560.12   483.7 1540.67
   493.6 1537.13     498  1536.5   503.5 1535.72     513 1536.85   552.8 1551.29
   562.7 1555.92   602.2 1578.69   612.1 1584.08     622 1588.22   711.3 1620.41
   741.1 1627.12   770.9 1636.49   820.5 1658.67   919.8 1695.11   959.4 1707.76
  1009.1 1720.77  1028.9 1727.42  1058.7 1739.84  1078.6 1750.07  1108.3  1766.7
#Mann= 3 , 0 , 0
       0      .1       0     498    .045       0     513      .1       0
Bank Sta=498,513
XS Rating Curve= 0 ,0
Exp/Cntr=0.3,0.1

Type RM Length L Ch R = 1 ,8864.2  ,310.1,300.4,292.4
XS GIS Cut Line= 3
     1937817.739      355364.496     1937516.823      355009.955
     1937309.251      354373.561
#Sta/Elev= 30
       0  1593.9    69.3 1592.18   118.7 1592.01   197.9 1593.24   286.9 1591.31
   366.1 1591.96   405.7 1591.24   415.6 1590.12   425.4  1587.7   435.3 1584.21
     465 1573.56     485 1565.46     505 1556.44     535 1541.73   574.9 1519.87
   584.9 1515.94   594.9 1515.04   599.9 1515.82   604.9  1516.6   694.8 1540.64
   704.8 1543.83   794.7  1585.2   844.7 1607.51   884.6 1621.54   944.6 1640.52
   964.6 1644.14   974.6 1644.73  1054.5 1640.82  1114.4 1641.07  1134.4 1639.06
#Mann= 3 , 0 , 0
       0      .1       0   584.9    .045       0   599.9      .1       0
Bank Sta=584.9,599.9
XS Rating Curve= 0 ,0
Exp/Cntr=0.3,0.1

Type RM Length L Ch R = 1 ,8563.9  ,284,291.7,297.7
XS GIS Cut Line= 3
     1938113.647      355165.279     1937738.133      354764.459
     1937384.266      354328.767
#Sta/Elev= 30
       0 1618.37   109.8 1605.08   189.7  1592.5   209.7 1590.15   229.7 1589.32
   329.6 1590.14   339.5 1587.52   349.5 1581.53   369.5 1561.09   379.5 1552.99
   389.5 1548.12   439.4 1542.31   459.4 1538.42   469.4 1534.44   489.3  1523.5
   529.3 1496.15   539.3 1492.16   541.7 1492.03   549.2 1491.62   556.7 1492.79
   618.2 1503.24   657.6 1514.87   677.3 1517.93   726.5 1530.18   805.3 1555.65
   864.4 1576.74   893.9 1583.85   913.6 1587.47  1021.9 1601.81  1110.5 1607.53
#Mann= 3 , 0 , 0
       0      .1       0   541.7    .045       0   556.7      .1       0
Bank Sta=541.7,556.7
XS Rating Curve= 0 ,0
Exp/Cntr=0.3,0.1

Type RM Length L Ch R = 1 ,8272    ,322,309.5,297
XS GIS Cut Line= 3
     1938184.901      355116.255     1937898.933      354447.708
     1937649.208       354136.17
#Sta/Elev= 30
       0 1634.17    49.8 1627.66   129.5 1621.18   149.4 1618.57   199.2 1606.58
   239.1  1595.9   278.9 1580.09   348.6 1559.49   378.5 1552.67   448.2 1540.72
   458.2 1537.41   468.2 1531.92   527.9 1487.14   537.9 1480.44   540.6 1479.56
   547.8 1477.21   555.6 1478.06   567.8 1482.52   607.6 1501.39   687.3 1533.94
   767.1  1571.2     787 1581.99   886.8 1643.86   896.8 1649.02   906.8 1652.99
   926.8 1656.75   946.7 1658.14  1026.6  1659.6  1096.5 1663.96  1126.4 1662.91
#Mann= 3 , 0 , 0
       0      .1       0   540.6    .045       0   555.6      .1       0
Bank Sta=540.6,555.6
XS Rating Curve= 0 ,0
Exp/Cntr=0.3,0.1

Type RM Length L Ch R = 1 ,7962.2  ,286.3,298.4,314.4
XS GIS Cut Line= 3
     1938554.112      354827.477      1938251.93      354462.265
     1937710.256      354079.065
#Sta/Elev= 30
       0  1672.5    98.8 1647.97   227.1 1612.78   266.6 1602.96   276.5 1599.37
   444.4 1525.76   464.1    1518   493.8 1508.77   503.7 1504.46     573 1464.58
   585.6 1458.65   592.9 1456.69   600.6 1457.44   602.8 1457.65   612.7 1462.54
   642.4 1481.54   701.8 1514.55   731.5 1535.87   800.8 1588.91   820.6 1602.74
   919.7 1656.32   939.5    1666   959.3 1674.27   979.1 1680.89   998.9  1685.8
  1018.7 1689.19  1068.2 1694.32  1097.9 1699.14  1117.7 1699.06  1137.5  1695.8
#Mann= 3 , 0 , 0
       0      .1       0   585.6    .045       0   600.6      .1       0
Bank Sta=585.6,600.6
XS Rating Curve= 0 ,0
Exp/Cntr=0.3,0.1

Type RM Length L Ch R = 1 ,7663.9  ,292.6,300.3,304.2
XS GIS Cut Line= 3
     1938619.728      354778.155      1938368.58      354202.725
     1938241.236      353686.688
#Sta/Elev= 30
       0 1660.39   239.2  1593.4     289  1570.2   368.7 1529.22   408.6  1511.5
   448.5  1498.8   508.3 1493.16   528.2 1488.67   558.1 1476.15   607.9 1447.32
   617.9 1444.04   620.3 1444.29   627.8 1445.06   635.3 1449.63   696.8 1500.03
   795.2  1569.5     805 1578.94   834.6 1613.82   854.2  1630.1   883.8 1651.52
   923.1 1673.23   982.2 1698.64  1001.9 1703.78  1041.2 1709.76  1051.1 1714.06
  1060.9 1722.79  1070.8 1735.97  1080.6 1745.33  1129.8 1762.48  1159.4 1770.58
#Mann= 3 , 0 , 0
       0      .1       0   620.3    .045       0   635.3      .1       0
Bank Sta=620.3,635.3
XS Rating Curve= 0 ,0
Exp/Cntr=0.3,0.1

Type RM Length L Ch R = 1 ,7363.9  ,294.2,296.8,299.4
XS GIS Cut Line= 3
     1938703.101       354766.71     1938665.694      354207.776
     1938629.758      353650.645
#Sta/Elev= 30
       0 1653.15      50 1635.75   230.1 1569.45   310.1  1536.3   330.1 1525.12
   360.1 1502.96   400.1  1475.8   430.1 1454.31   440.1  1448.6   450.2  1444.6
   470.2 1439.18   490.2 1436.07   510.2 1435.01   552.7 1435.02   560.2 1434.77
   567.7  1435.2   580.1 1438.84   590.1 1445.29   649.9 1489.29   689.8 1521.93
   699.8 1527.62   709.7 1531.48   779.5 1552.31   839.3 1575.92   909.1 1601.06
     939 1613.89     959 1620.46   978.9 1624.46  1078.6 1638.54  1118.5 1640.26
#Mann= 3 , 0 , 0
       0      .1       0   552.7    .045       0   567.7      .1       0
Bank Sta=552.7,567.7
XS Rating Curve= 0 ,0
Exp/Cntr=0.3,0.1

Type RM Length L Ch R = 1 ,7066.7  ,317.6,290.1,262.5
XS GIS Cut Line= 3
      1938936.49      354760.822     1938965.201      354136.562
     1938712.528      353642.258
#Sta/Elev= 30
       0 1637.98    69.4 1613.67   138.9 1600.38   218.2 1582.13     248 1573.87
   287.7 1560.12   317.4 1546.23   337.3 1534.94   386.9 1502.04   436.4 1466.66
   456.3  1454.4   505.9 1428.37   515.8 1424.28   521.7 1423.87   525.7  1423.6
   536.7 1426.91   565.4 1438.02   674.5 1475.08   714.1 1490.74   773.6  1524.4
   862.8 1581.35   892.6 1599.06   932.2 1619.49     962  1631.8  1001.6 1645.12
  1031.4 1651.77  1051.2 1653.18  1110.7 1652.72  1160.2 1655.25  1180.1 1658.94
#Mann= 3 , 0 , 0
       0      .1       0   521.7    .045       0   536.7      .1       0
Bank Sta=521.7,536.7
XS Rating Curve= 0 ,0
Exp/Cntr=0.3,0.1

Type RM Length L Ch R = 1 ,6776.5  ,323.3,319.9,316.4
XS GIS Cut Line= 3
     1939680.301      354312.629     1939056.179      354047.403
     1938778.079      353602.927
#Sta/Elev= 30
       0    1636    39.9 1637.92   109.7 1638.14   129.6 1635.85   149.6 1629.57
   169.5 1619.23   229.4 1579.11   279.2  1551.4     379 1504.78   428.8 1478.47
   468.7 1450.51   478.7 1441.63   498.6 1419.89   508.6  1412.8   520.7 1409.49
   528.6 1408.68   535.7 1408.81   578.4 1413.69   618.3 1423.23   648.2 1434.71
   707.8 1463.04   757.3 1484.88   866.1 1556.95  1004.6  1653.2  1034.3 1671.11
    1064 1686.32  1083.7 1693.64  1123.3 1700.14    1153 1701.65  1202.4  1700.3
#Mann= 3 , 0 , 0
       0      .1       0   520.7    .045       0   535.7      .1       0
Bank Sta=520.7,535.7
XS Rating Curve= 0 ,0
Exp/Cntr=0.3,0.1

Type RM Length L Ch R = 1 ,6456.7  ,287.6,292.7,298.9
XS GIS Cut Line= 3
     1939860.855      353955.857     1939185.369      353789.024
     1938823.833      353533.845
#Sta/Elev= 30
       0 1566.54    59.6  1545.6   109.3 1520.99     169 1494.18   228.6  1460.7
   238.6 1457.04   258.4 1453.63   318.1 1451.62   407.5 1450.56   427.4 1447.93
   447.3 1440.84   467.2 1431.57   526.8    1399   531.8 1397.61   536.8 1396.22
   546.8 1397.08   646.1 1436.18   675.9 1450.03   705.6 1466.32   774.4 1510.54
     804 1530.63   843.3 1558.75   902.3 1603.78   951.5 1637.45  1000.6 1673.74
    1040 1698.91  1049.8 1703.91  1059.6 1707.25  1069.5 1708.63  1138.3 1707.58
#Mann= 3 , 0 , 0
       0      .1       0   531.8    .045       0   546.8      .1       0
Bank Sta=531.8,546.8
XS Rating Curve= 0 ,0
Exp/Cntr=0.3,0.1

Type RM Length L Ch R = 1 ,6163.9  ,291.4,299.9,309.9
XS GIS Cut Line= 3
     1939929.141      353813.468     1939438.784      353571.902
     1938955.354      353303.012
#Sta/Elev= 30
       0 1611.01    39.8  1602.6    59.6 1597.41   119.3 1579.96   139.1 1572.23
   188.8 1548.58   208.7 1538.32   228.6 1524.62   258.4 1507.75   298.2 1482.68
     318 1472.53   357.8 1457.87   437.3 1434.76   457.2 1427.97   516.8 1398.41
   536.7 1387.71   539.1 1387.06   546.6 1385.02   554.1 1385.12   566.4 1387.94
   615.8  1413.6   694.8 1459.24   744.2 1490.79   773.8 1508.33   892.4 1572.95
   912.1 1585.26   931.9 1598.92  1030.7 1670.48  1050.4 1682.25  1099.8    1707
#Mann= 3 , 0 , 0
       0      .1       0   539.1    .045       0   554.1      .1       0
Bank Sta=539.1,554.1
XS Rating Curve= 0 ,0
Exp/Cntr=0.3,0.1

Type RM Length L Ch R = 1 ,5863.9  ,298.4,299.9,295.4
XS GIS Cut Line= 3
     1939981.982      353743.437     1939608.385      353333.066
     1939293.797       352888.92
#Sta/Elev= 30
       0 1611.46    49.6 1590.71    99.1 1567.84   237.8 1499.86   317.1 1459.88
   346.8 1445.45   376.6 1431.98   396.4 1423.92   416.2 1416.65   485.6 1393.34
   515.3 1383.89   535.1 1376.63     545  1373.4   547.5 1373.18     555 1372.52
   562.5 1373.53   564.8 1373.84   574.8 1378.46   604.4 1397.07   683.6 1453.17
   752.9 1498.18   792.5 1525.44   822.2 1547.34   940.9 1638.73   960.7 1654.41
  1010.2 1696.18  1020.1 1703.98    1030 1710.78  1039.9 1715.91  1099.2 1740.82
#Mann= 3 , 0 , 0
       0      .1       0   547.5    .045       0   562.5      .1       0
Bank Sta=547.5,562.5
XS Rating Curve= 0 ,0
Exp/Cntr=0.3,0.1

Type RM Length L Ch R = 1 ,5563.9  ,314.3,299.9,291.6
XS GIS Cut Line= 3
     1940191.118       353585.24     1939852.622      353159.343
     1939446.642      352778.019
#Sta/Elev= 30
       0 1616.18    69.2 1584.04   138.5 1556.51   158.3  1547.9   197.8 1526.73
   257.2 1492.92   346.2 1449.63   395.7  1422.6   464.9 1386.07   484.7 1377.72
   494.6 1374.28   524.2 1366.01   536.5 1363.31     544 1362.51   551.5  1363.5
     554 1363.83   573.9 1371.31   623.6 1387.05   633.5 1390.71   752.9  1445.8
   822.5 1481.62   902.1  1519.4   931.9 1534.58   971.7 1557.26   991.6 1569.97
  1011.5 1583.87  1021.4 1588.32  1041.3 1595.38  1051.3 1599.64    1101 1623.39
#Mann= 3 , 0 , 0
       0      .1       0   536.5    .045       0   551.5      .1       0
Bank Sta=536.5,551.5
XS Rating Curve= 0 ,0
Exp/Cntr=0.3,0.1

Type RM Length L Ch R = 1 ,5263.9  ,407.5,427.5,444.8
XS GIS Cut Line= 3
     1940538.396      353058.321     1940013.883      352916.563
     1939493.964      352705.512
#Sta/Elev= 30
       0 1644.93    69.2 1609.01   138.3 1570.77   197.6 1536.22   276.6 1488.77
   316.1 1466.55   365.5 1440.82   434.7 1410.63   444.5 1405.32   454.4 1398.32
   474.2 1382.48   493.9 1369.77   523.6 1354.66   535.8 1351.24   543.3 1350.68
   550.8 1351.19   651.6 1362.16   661.5 1363.92   681.2 1371.07   730.4 1393.54
     819 1436.61   858.4 1460.08   907.6 1482.73   937.1 1501.28   986.3 1530.16
  1025.7  1551.8  1045.4 1558.03  1084.8 1567.15  1094.6 1571.29  1104.4 1577.37
#Mann= 3 , 0 , 0
       0      .1       0   535.8    .045       0   550.8      .1       0
Bank Sta=535.8,550.8
XS Rating Curve= 0 ,0
Exp/Cntr=0.3,0.1

Type RM Length L Ch R = 1 ,4836.3  ,230,218.8,207.7
XS GIS Cut Line= 2
     1940286.209      352913.811     1940007.814      352289.698
#Sta/Elev= 30
       0 1482.53    29.7 1471.76    59.4  1459.7    89.1 1445.75     109 1434.81
   128.8 1422.31   178.3 1386.73   188.2 1380.28     208 1369.19   237.7 1356.96
   267.4 1347.85   297.1 1342.09   326.8 1339.34   396.2 1336.09   419.1 1330.87
   425.9 1329.22   434.1 1329.02   435.8 1328.98   445.7 1332.39   475.4 1347.21
   485.3 1353.04   495.2  1359.7   534.8 1389.25   554.6 1401.44   574.4 1410.65
   594.2 1417.98   643.8 1431.78   653.7 1435.97   673.5 1447.95   683.4 1452.68
#Mann= 3 , 0 , 0
       0      .1       0   419.1    .045       0   434.1      .1       0
Bank Sta=419.1,434.1
XS Rating Curve= 0 ,0
Exp/Cntr=0.3,0.1

Type RM Length L Ch R = 1 ,4617    ,251.4,253.1,251.6
XS GIS Cut Line= 3
     1940721.784      352776.743      1940153.38      352333.368
     1939934.873      352007.577
#Sta/Elev= 30
       0 1642.06      20  1634.5      30 1629.47    50.1 1617.34   100.1 1580.93
   150.2 1547.24   210.3 1500.56   240.3 1478.98   260.3 1465.83   290.4  1448.2
   330.4  1427.1   370.4 1411.26   390.5 1401.94   400.5 1394.86   430.5 1370.39
   480.6 1334.58   530.6 1311.21   535.6  1310.4   540.7 1309.58   550.6 1310.24
   560.7 1313.18   630.8 1339.97   680.8 1363.89   720.9 1381.65   789.5 1406.79
   828.8 1418.97     917  1453.6   995.5 1482.33  1093.6 1513.39  1113.2 1520.48
#Mann= 3 , 0 , 0
       0      .1       0   535.6    .045       0   550.6      .1       0
Bank Sta=535.6,550.6
XS Rating Curve= 0 ,0
Exp/Cntr=0.3,0.1
